--- LeadmineRun.prj (project) ---

Proj Title=LeadmineRun
Current Plan=p01
Default Exp/Contr=0.3,0.1
SI Units
Geom File=g01
Flow File=f01
Plan File=p01
Y Axis Title=Elevation
X Axis Title(PF)=Main Channel Distance
X Axis Title(XS)=Station
BEGIN DESCRIPTION:
September 2018
Tucker County ABFE Study
US Army Corps of Engineers, Pittsburgh District
NAD 1983 UTM 17N (meters)
END DESCRIPTION:
DSS Export Rating Curves= 0
DSS Export Rating Curve Sorted= 0
DSS Export Volume Flow Curves= 0
DXF OffsetX= 0
DXF OffsetY= 0
DXF ScaleX= 1
DXF ScaleY= 10

--- LeadmineRun.p01 (plan) ---

Plan Title=LeadmineRun_plan
Program Version=5.05
Short Identifier=Plan1_subcritical
Geom File=g01
Flow File=f01
Subcritical Flow
K Sum by GR= 0
Std Step Tol= 0.003
Critical Tol= 0.003
Num of Std Step Trials= 20
Max Error Tol= 0.1
Flow Tol Ratio= 0.001
Split Flow NTrial= 30
Split Flow Tol= 0.006
Split Flow Ratio= 0.02
Log Output Level= 0
Friction Slope Method= 1
Unsteady Friction Slope Method= 2
Unsteady Bridges Friction Slope Method= 1
Parabolic Critical Depth
Global Vel Dist= 0 , 0 , 0
Global Log Level= 0
CheckData=True
Encroach Param=-1 ,0,0, 0
Computation Interval=1MIN
Output Interval=1HOUR
Instantaneous Interval=1HOUR
Mapping Interval=1HOUR
Computation Time Step Use Courant=        0
Computation Time Step Use Time Series=    0
Computation Time Step Count To Double=0
Computation Time Step Max Doubling=0
Computation Time Step Max Halving=0
Computation Time Step Residence Courant=0
Run HTab= 0
Run UNet= 0
Run Sediment= 0
Run PostProcess= 0
Run WQNet= 0
Run RASMapper=-1
UNET Theta= 1
UNET Theta Warmup= 1
UNET ZTol= 0.006
UNET ZSATol= 0.006
UNET MxIter= 20
UNET Max Iter WO Improvement= 0
UNET MaxInSteps= 0
UNET DtIC= 0
UNET DtMin= 0
UNET MaxCRTS= 20
UNET WFStab= 2
UNET SFStab= 1
UNET WFX= 1
UNET SFX= 1
UNET 1D Methodology=Finite Difference
UNET DSS MLevel= 4
UNET Pardiso=0
UNET DZMax Abort= 30
UNET Use Existing IB Tables=-1
UNET Froude Reduction=False
UNET Froude Limit= 0.8
UNET Froude Power= 4
UNET D1 Cores= 0
UNET D2 Coriolis=0
UNET D2 Cores= 0
UNET D2 Theta= 1
UNET D2 Theta Warmup= 1
UNET D2 Z Tol= 0.003
UNET D2 Volume Tol= 0.003
UNET D2 Max Iterations= 20
UNET D2 Equation= 0
UNET D2 RampUpFraction=0.1
UNET D2 TimeSlices= 1
UNET D2 BCVolumeCheck=0
UNET D1D2 MaxIter= 0
UNET D1D2 ZTol=0.003
UNET D1D2 QTol=0.1
UNET D1D2 MinQTol=0.03
Write IC File= 0
Write IC File at Fixed DateTime=0
Write IC File at Sim End=0
Echo Input=False
Echo Parameters=False
Echo Output=False
Write Detailed= 0
HDF Write Warmup=0
HDF Write Time Slices=0
HDF Flush=0
HDF Face Node Velocities=0
HDF Compression= 1
HDF Chunk Size= 1
HDF Spatial Parts= 1
HDF Use Max Rows=0
HDF Fixed Rows= 1
Calibration Method= 0
Calibration Iterations= 20
Calibration Max Change=0.05
Calibration Tolerance=0.2
Calibration Maximum=1.5
Calibration Minimum=0.5
Calibration Optimization Method= 1
WQ AD Non Conservative
WQ ULTIMATE=-1
WQ Max Comp Step=1HOUR
WQ Output Interval=15MIN
WQ Output Selected Increments= 0
WQ Output face flow=0
WQ Output face velocity=0
WQ Output face area=0
WQ Output face dispersion=0
WQ Output cell volume=0
WQ Output cell surface area=0
WQ Output cell continuity=0
WQ Output cumulative cell continuity=0
WQ Output face conc=0
WQ Output face dconc_dx=0
WQ Output face courant=0
WQ Output face peclet=0
WQ Output face adv mass=0
WQ Output face disp mass=0
WQ Output cell mass=0
WQ Output cell source sink temp=0
WQ Output nsm pathways=0
WQ Output nsm derived pathways=0
WQ Output MaxMinRange=-1
WQ Daily Max Min Mean=-1
WQ Daily Range=0
WQ Daily Time=0
WQ Create Restart=0
WQ Fixed Restart=0
WQ System Summary=0
WQ Write To DSS=0
WQ Use Fixed Temperature=0
Sorting and Armoring Iterations= 10
XS Update Threshold= 0.02
Bed Roughness Predictor= 0
Hydraulics Update Threshold= 0.02
Energy Slope Method= 1
Volume Change Method= 1
Sediment Retention Method= 0
XS Weighting Method= 0
Number of US Weighted Cross Sections= 1
Number of DS Weighted Cross Sections= 1
Upstream XS Weight=0
Main XS Weight=1
Downstream XS Weight=0
Number of DS XS's Weighted with US Boundary= 1
Upstream Boundary Weight= 1
Weight of XSs Associated with US Boundary= 0
Number of US XS's Weighted with DS Boundary= 1
Downstream Boundary Weight= 0.5
Weight of XSs Associated with DS Boundary= 0.5
Percentile Method= 0
Sediment Output Level= 4
Mass or Volume Output= 0
Output Increment Type= 1
Profile and TS Output Increment= 1
XS Output Flag= 0
XS Output Increment= 10
Write Gradation File= 0
Read Gradation Hotstart= 0
Write HDF5 File= 1
Write Binary Output= 1
Write DSS Sediment File= 0
SV Curve= 0
Specific Gage Flag= 0

--- LeadmineRun.f01 (steady flow) ---

Flow Title=LeadmineRun_flow
Program Version=5.05
Number of Profiles= 1
Profile Names=PF 1
River Rch & RM=Leadmine Run,1               ,6675.083
   14.64
River Rch & RM=Leadmine Run,1               ,5760.72
 17.7262
River Rch & RM=Leadmine Run,1               ,4571.733
 20.8693
River Rch & RM=Leadmine Run,1               ,4023.36
 21.4356
River Rch & RM=Leadmine Run,1               ,3017.46
 31.3181
River Rch & RM=Leadmine Run,1               ,2926.037
 31.3748
River Rch & RM=Leadmine Run,1               ,1554.48
 34.5462
River Rch & RM=Leadmine Run,1               ,457.2
 35.8488
River Rch & RM=Leadmine Run,1               ,91.44003
  36.047
Boundary for River Rch & Prof#=Leadmine Run,1               , 1
Up Type= 2
Dn Type= 1
Dn Known WS=562.05
DSS Import GetInterval= 0
DSS Import GetPeak= 0
DSS Import FillOption= 0

--- LeadmineRun.g01 (geometry) ---

Geom Title=LeadmineRun_geometry
Program Version=5.05

River Reach=Leadmine Run    ,1
Reach XY= 30
     627062.6643    4341808.6917      626828.235     4341953.551
     626389.0464    4342037.3771     626322.7766    4342103.5726
     626085.4765    4342094.7372     625873.8094    4341928.0493
     625785.3943    4341766.3004625646.2254128054341651.30033598
625502.8702167694341345.22992561625355.2526126054341201.54678234
     625303.3666    4340842.1972     625361.1389    4340273.5061
625240.8868384144340196.92417637     625317.6541    4339979.6538
      625247.804    4339926.2078     625000.2978    4339942.2272
     624930.3034    4339993.9413     624794.0427    4340022.7809
     624717.9559    4340120.8092     624743.9336    4340205.4958
     624609.6277    4340332.2118624367.5486216454340402.64286204
     623911.1263    4340744.9626     623779.8927    4340759.7793
     623711.1009    4340825.9253      623551.941    4340853.4549
623224.2166256094341209.01565518623226.1264399414341251.07236509
     623104.0573    4341288.9471      623094.282    4341337.5076

Type RM Length L Ch R = 1 ,6675.083,92.37,91.36,87.89
XS GIS Cut Line= 3
     627010.9928    4341755.4983     627023.7628    4341829.3562
     627073.4346     4341931.182
#Sta/Elev= 30
       0   756.8       6   753.4   11.99  749.61   14.99  749.24   17.99  747.47
   29.98  738.78   35.98  735.37   38.98  734.15   44.97  733.11   53.97   731.1
   56.96  730.16   62.96  726.75   65.96  726.08   71.96  726.72   81.08  727.01
   90.26  727.03   96.39  726.63   99.45  726.79  105.57  727.47  108.64  728.63
  117.82  732.94  133.13  738.96  136.19  739.06  154.57  745.59  163.75  748.47
  166.81  748.41  169.88  749.03  179.06   751.7  182.12  753.04  188.25  756.26
#Mann= 3 , 0 , 0
       0      .1       0   62.96      .1       0   99.45      .1       0
Bank Sta=62.96,99.45
XS Rating Curve= 0 ,0
Exp/Cntr=0.3,0.1

Type RM Length L Ch R = 1 ,6583.727,92.73,91.44,85.95
XS GIS Cut Line= 3
      626913.626     4341802.065     626947.7868    4341873.6562
     627005.7011     4341975.632
#Sta/Elev= 30
       0  757.36     6.1  753.86    9.15   752.5    12.2  752.32   15.25  751.24
   24.41  746.68   39.66  738.57   42.71  738.21   45.76     737   54.92  731.45
   64.07  725.02   67.12  723.19   70.17  721.97   76.27  721.45   79.32  721.48
   82.33  721.93   97.37  723.82  109.39  724.93  118.42  726.16  127.44  728.07
  133.45  730.74  139.46  732.34  145.48  735.09  151.49  739.05  163.52  744.95
  166.53  746.09  169.53  746.45  178.56  750.15  184.57  753.09   196.6  757.48
#Mann= 3 , 0 , 0
       0      .1       0   70.17      .1       0   82.33      .1       0
Bank Sta=70.17,82.33
XS Rating Curve= 0 ,0
Exp/Cntr=0.3,0.1

Type RM Length L Ch R = 1 ,6492.291,89.76,91.54,99.49
XS GIS Cut Line= 3
     626796.1507    4341846.5151     626878.7224    4341925.5823
     627002.5261     4342101.574
#Sta/Elev= 30
       0  746.92    6.02   744.9   18.05  742.29   42.12  730.45   48.14  726.81
   51.14  726.59   66.19  728.93    72.2  728.69   81.23  726.47   93.26  721.78
   99.28  718.73  102.29  718.52  111.31  718.99  135.84  719.98  148.14  721.68
  163.51   726.2  178.88  732.27  191.17  736.31  203.47  739.52  212.69  740.96
  224.98  740.83  231.13  741.74  234.21  741.36  243.43  742.26  277.24  740.39
  286.46  740.55  295.68  741.66  301.83  743.45  323.35  747.11   329.5   748.9
#Mann= 3 , 0 , 0
       0      .1       0   99.28      .1       0  111.31      .1       0
Bank Sta=99.28,111.31
XS Rating Curve= 0 ,0
Exp/Cntr=0.3,0.1

Type RM Length L Ch R = 1 ,6400.754,90.61,91.59,88.65
XS GIS Cut Line= 3
      626774.984    4341858.1568     626792.5007    4341949.7002
     626801.4424    4342047.5989
#Sta/Elev= 30
       0  747.16    6.01  746.18   24.05  740.75   33.07  736.99   36.08   736.8
   42.09  733.72   51.11  727.84   60.13  723.36   66.14  721.83   69.15  720.46
   72.16  719.46   78.17  717.79   84.18   716.6   99.79  715.22  105.49  714.68
  108.56   714.8  111.64  715.29  117.78  716.33  120.85   717.2  123.92  717.49
  133.14  723.37  139.29  726.55  151.57  733.66  154.65  733.85  160.79  737.41
  163.86  738.84  166.93   739.9  179.22  742.79  182.29  742.83  191.51  746.84
#Mann= 3 , 0 , 0
       0      .1       0   99.79      .1       0  111.64      .1       0
Bank Sta=99.79,111.64
XS Rating Curve= 0 ,0
Exp/Cntr=0.3,0.1

Type RM Length L Ch R = 1 ,6309.168,91.79,90.62,89.35
XS GIS Cut Line= 3
     626686.0838    4341896.2569     626704.6459    4341965.6618
     626739.0006    4342063.4739
#Sta/Elev= 30
       0  747.11    5.99  743.54    8.98  742.93   11.97  741.72   23.95  734.09
   35.92  726.16   38.92  726.03   41.91  723.81    47.9  717.88   50.89  715.28
   53.88  713.34   56.88  712.56   71.84  712.93   77.94  712.89   84.04  712.53
   90.14  712.93   99.29  713.69  102.34  714.32  105.38  715.61  114.53  720.57
  123.68  724.81  126.73  725.85  129.78  726.22  135.88  728.81  141.97  731.68
  145.02  733.74  154.17  738.45  160.27   740.3  169.42  745.07  175.51  747.76
#Mann= 3 , 0 , 0
       0      .1       0   56.88      .1       0   90.14      .1       0
Bank Sta=56.88,90.14
XS Rating Curve= 0 ,0
Exp/Cntr=0.3,0.1

Type RM Length L Ch R = 1 ,6218.55 ,90.02,91.1,96.15
XS GIS Cut Line= 2
      626587.835    4341923.3106      626669.856    4342107.1964
#Sta/Elev= 30
       0  745.95   24.41  733.71   27.46  733.08   33.56  730.88   54.91  722.21
   57.96  721.87   61.01  720.45   64.07  717.67   67.12  714.52   70.17  712.86
   79.32  710.07   82.37  709.43   88.47  709.72   91.52  710.43   94.57  710.69
  103.73  710.59  122.03     711  125.08  711.91  131.18   715.1  134.23  716.28
  140.33  718.06  143.38  719.51  146.44  721.48  149.49   721.9  155.59  725.41
  170.84  732.96  176.94  735.29  179.99  735.56  189.15  740.27  201.35  747.31
#Mann= 3 , 0 , 0
       0      .1       0   79.32      .1       0   88.47      .1       0
Bank Sta=79.32,88.47
XS Rating Curve= 0 ,0
Exp/Cntr=0.3,0.1

Type RM Length L Ch R = 1 ,6127.446,91.96,92.41,92.55
XS GIS Cut Line= 2
     626526.9807    4341945.8002     626550.7933    4342149.5298
#Sta/Elev= 30
       0  747.17    3.06  745.47    9.18  742.57   12.25  742.42   15.31  741.11
   30.61  733.96   36.74  730.35    39.8  729.71   42.86  728.23   55.11  719.65
   67.35  710.57   70.41  709.85   73.47  708.23   76.54  706.97    79.6  706.94
   84.05  707.43   97.97  708.36  131.64  709.57   134.7  710.28  137.76  711.61
  143.89  715.01  156.13  722.85  159.19  724.18  162.26  724.93  171.44  730.76
  177.56  734.01  183.69  737.18  186.75  738.36  189.81  738.79  205.12   746.7
#Mann= 3 , 0 , 0
       0      .1       0   76.54      .1       0   84.05      .1       0
Bank Sta=76.54,84.05
XS Rating Curve= 0 ,0
Exp/Cntr=0.3,0.1

Type RM Length L Ch R = 1 ,6035.04 ,94.98,91.44,79.41
XS GIS Cut Line= 4
     626451.5743    4341939.1856      626444.182    4342030.6541
     626445.1264    4342046.4727     626468.7723    4342186.5715
#Sta/Elev= 30
       0  747.44    9.18  742.71   18.35  736.24   24.47     733   27.53  731.75
   33.65  730.44   45.88  726.41   55.06  722.52   58.12  721.95   61.18  720.35
    67.3  713.97   73.41  708.35   76.47  706.16   79.53  705.23   94.41  704.92
   99.69   705.2  116.68  706.44  140.87  705.93  149.94  706.35  155.98  707.53
  168.07  713.97  177.14  717.28  180.17  717.85  183.19   719.2  204.35  730.29
   210.4  731.89  219.46   735.6  234.58  740.49  240.62  741.74  249.69  746.01
#Mann= 3 , 0 , 0
       0      .1       0   79.53      .1       0   99.69      .1       0
Bank Sta=79.53,99.69
XS Rating Curve= 0 ,0
Exp/Cntr=0.3,0.1

Type RM Length L Ch R = 1 ,5943.6  ,27.83,26.41,20.87
XS GIS Cut Line= 4
      626341.772     4341949.769     626348.1311    4342040.1884
      626380.477    4342088.6501     626388.0742    4342181.2799
#Sta/Elev= 30
       0  738.29    3.02  736.86    6.04  736.57   12.09  733.54   30.21  725.43
   33.24  725.42   36.26  724.07    42.3   720.9   57.41  711.52   60.43  710.04
   63.45  709.81   78.56   704.2   81.58  703.33   87.62  702.73   90.64  702.35
   96.78  702.27   99.84  702.69  105.98  703.55  127.44  704.78   166.9  705.37
  172.89  706.05  178.89  708.38  184.88  711.45  187.88  711.55  202.87  719.02
  214.87  726.02  217.86  726.42  220.86   727.6  232.85  733.49  241.85  738.72
#Mann= 3 , 0 , 0
       0      .1       0   87.62      .1       0   99.84      .1       0
Bank Sta=87.62,99.84
XS Rating Curve= 0 ,0
Exp/Cntr=0.3,0.1

Type RM Length L Ch R = 1 ,5917.195,19.6,51.47,54.92
XS GIS Cut Line= 6
     626324.6517    4341952.8432     626326.7684    4342056.0309
     626333.9783    4342071.4429     626348.8611    4342078.3882
      626358.783    4342093.9325     626366.0591    4342182.8989
#Sta/Elev= 30
       0     736    6.07  734.47   30.36  724.42   33.39  724.31   39.46  721.71
   45.53  718.39   48.57  716.16   54.64   710.4   57.68  707.82   60.71  705.82
   63.75  705.75   69.82  703.25   72.85  702.51   81.96  701.62   88.03  701.02
    94.1  701.25  100.17  701.98  122.96  702.49  139.72  701.92  148.94  702.08
  164.02  703.38  169.97  704.65  172.94  705.66  187.82  712.11  190.79  712.49
  193.77   713.4  217.57  724.79  220.55  725.81  223.52  726.31  244.35  736.86
#Mann= 3 , 0 , 0
       0      .1       0   81.96      .1       0  148.94      .1       0
Bank Sta=81.96,148.94
XS Rating Curve= 0 ,0
Exp/Cntr=0.3,0.1

Type RM Length L Ch R = 1 ,5865.723,12.05,13.56,14.01
XS GIS Cut Line= 6
     626311.8326    4341952.9358     626314.4996    4342063.9834
     626310.5838    4342087.5843     626306.7738     4342105.576
     626306.8796    4342113.5135     626321.6302    4342191.5049
#Sta/Elev= 30
       0     735       3  733.95       6  733.72   15.01  730.43   33.02  723.02
   36.03  723.02   42.03  720.54   45.03  719.01   48.03  717.04   51.04  714.49
   57.04  708.61   60.04  705.99   63.05  705.26   69.05  703.07   81.06  701.24
   87.06  700.81   99.07  701.33     135   701.6   144.2  701.24  150.33  700.47
  156.04  700.88   176.6  708.72   182.7   711.5  188.81  712.95  210.18  724.13
  213.23  725.52  216.28  725.66  225.44  729.76   234.6  734.81  240.71  737.64
#Mann= 3 , 0 , 0
       0      .1       0   81.06      .1       0  156.04      .1       0
Bank Sta=81.06,156.04
XS Rating Curve= 0 ,0
Exp/Cntr=0.3,0.1

Type RM Length L Ch R = 1 ,5852.16 ,36.14,29.8,28.98
XS GIS Cut Line= 4
     626304.7303    4341947.1231     626305.3458    4342053.3359
     626293.2721    4342102.9726     626282.2407    4342214.3528
#Sta/Elev= 30
       0  737.47    6.07   734.4     9.1  733.42   12.14  733.04   21.24  729.78
   36.42  723.49   39.45  722.62   42.49   722.4   45.52  721.16   54.62  715.94
   66.76  704.75    69.8  703.21   72.83  703.17   84.97  701.03   88.01  700.56
   97.11  701.04  136.26  700.84  160.32  699.21  166.37  699.64  175.45   701.2
  178.47  702.09  184.52  706.33  190.57  709.38  199.65     712  211.75  716.89
  220.82  721.16  226.87  722.52  251.07  732.57  257.12  733.59  269.22  738.03
#Mann= 3 , 0 , 0
       0      .1       0   84.97      .1       0  166.37      .1       0
Bank Sta=84.97,166.37
XS Rating Curve= 0 ,0
Exp/Cntr=0.3,0.1

Type RM Length L Ch R = 1 ,5822.362,33.42,30.45,28.17
XS GIS Cut Line= 6
     626271.8443    4341943.7883      626259.938    4341974.8769
     626262.9146    4342039.6999     626266.7114    4342080.3532
     626259.5147    4342167.9834     626264.3831    4342216.0318
#Sta/Elev= 30
       0  734.37   15.13  727.26   18.16  726.22   24.21  725.13   33.29   720.7
   39.19  718.27   50.99  714.13   53.94  713.99   59.84  710.74   68.69  703.78
   71.64  702.76   77.53  701.85   98.18  700.01  104.01   699.7  109.85  700.39
  124.43  700.51  159.43  698.21  162.34  698.52  168.18  700.13  179.87  701.09
  182.81  702.05  191.64  707.07  200.47  710.45  206.36  711.43  229.99  719.73
     233  720.65  236.02  720.81  260.17  729.47  263.19  729.58  275.26  734.73
#Mann= 3 , 0 , 0
       0      .1       0   98.18      .1       0  162.34      .1       0
Bank Sta=98.18,162.34
XS Rating Curve= 0 ,0
Exp/Cntr=0.3,0.1

Type RM Length L Ch R = 1 ,5791.916,30.99,31.2,31.56
XS GIS Cut Line= 6
     626225.2246    4341935.1496     626222.2613    4341999.4964
     626233.4797    4342078.8716     626236.0197    4342100.8849
     626234.3263    4342151.4734     626241.9463    4342220.6885
#Sta/Elev= 30
       0  736.16    6.13  734.75   12.27  731.91   27.61  722.91   36.81  721.11
   46.01  718.22   58.28  711.98   61.35  711.06   70.35  709.92   76.29  708.07
   79.26  706.72    85.2  702.69   88.17  701.59   91.14  700.88  120.83  698.65
  138.64  699.16  155.66  697.96  159.99  698.41  166.74  699.47  186.94  700.59
  196.06  705.13   199.1  706.07  214.31  708.21  220.38  709.69  226.44  711.77
  241.58  718.92  250.66  721.39  268.82   729.7  274.88  730.64  286.99   734.5
#Mann= 3 , 0 , 0
       0      .1       0  120.83      .1       0  159.99      .1       0
Bank Sta=120.83,159.99
XS Rating Curve= 0 ,0
Exp/Cntr=0.3,0.1

Type RM Length L Ch R = 1 ,5760.72 ,85.45,91.44,94.45
XS GIS Cut Line= 4
      626179.053    4341929.9252     626203.1774    4342084.8693
     626204.3841    4342100.8132     626204.1884    4342216.9987
#Sta/Elev= 30
       0  729.78   12.06  726.05   18.09   725.2   42.22  717.17   48.25  716.32
   54.28  714.67   63.33  711.83   72.37  708.33   75.39  708.32   81.42   706.9
    96.5  701.31  102.53  699.92  105.55  699.71  114.59  697.98  123.64  697.25
  132.69  697.14  156.81  697.16  170.14  696.62  175.86  697.02  197.26   699.1
  209.49  703.45  218.66  705.84  224.78  706.74  249.24  716.88   252.3  717.91
  255.35  718.17  279.81  727.59  282.87  728.52  285.93  728.74  288.99  729.76
#Mann= 3 , 0 , 0
       0      .1       0  132.69      .1       0  175.86      .1       0
Bank Sta=132.69,175.86
XS Rating Curve= 0 ,0
Exp/Cntr=0.3,0.1

Type RM Length L Ch R = 1 ,5669.28 ,73.78,91.44,97.48
XS GIS Cut Line= 4
     626149.9487    4341920.6648     626116.2779    4342085.5907
     626112.9598    4342107.9125     626090.4174     4342195.832
#Sta/Elev= 30
       0  730.07    3.06  728.95   12.24   724.5   21.42  721.51   27.54  719.02
   33.67  717.75   42.85  714.82   58.15  712.06   64.27  711.59   85.69  707.69
   91.82  704.91   94.88  704.89   97.94  704.26  122.42  697.47  134.66   695.8
  153.03  694.77  168.33   694.9  188.07  694.16  193.92  694.42     203  695.54
  206.02  696.91   215.1  702.79  218.12  704.18  221.15  704.61  224.17  705.94
  233.25   710.6  248.38  717.57   251.4  718.02  266.53  724.85  281.66  729.57
#Mann= 3 , 0 , 0
       0      .1       0  153.03      .1       0  193.92      .1       0
Bank Sta=153.03,193.92
XS Rating Curve= 0 ,0
Exp/Cntr=0.3,0.1

Type RM Length L Ch R = 1 ,5577.84 ,99.47,91.44,88.81
XS GIS Cut Line= 6
      626128.782    4341910.0814     626077.2567    4342028.2006
     626050.0244    4342050.4601     626038.7827    4342055.7565
     626033.9744     4342058.962     625954.1567     4342129.686
#Sta/Elev= 30
       0  729.57   12.27  725.23   15.34  724.87   30.68  718.04   36.82  715.78
   49.09  712.36   52.16   712.2   55.23  711.51   70.57  707.49   82.84  705.42
   95.12  704.16  110.46  700.92   116.6     699  119.66  698.71  128.87     695
   131.8  694.37  149.39  693.13   171.5  692.16  188.34  691.91  191.39  692.19
  194.43  693.34  200.53  696.73  209.67  700.44  227.95  709.51     231  710.37
  234.04  710.52  261.47  720.26  279.75  726.03  285.84  727.13  288.89  728.38
#Mann= 3 , 0 , 0
       0      .1       0   171.5      .1       0  191.39      .1       0
Bank Sta=171.5,191.39
XS Rating Curve= 0 ,0
Exp/Cntr=0.3,0.1

Type RM Length L Ch R = 1 ,5486.4  ,90.86,91.44,89.39
XS GIS Cut Line= 6
     626055.4923    4341891.7369     625986.8219    4341975.6491
     625983.2698    4341983.7191     625979.0106    4341988.9804
     625974.5849    4341997.4772     625892.5086     4342078.004
#Sta/Elev= 30
       0  719.95   12.05  715.25   15.06  714.21   18.07  713.89    24.1  711.42
   42.17  705.32    51.2  703.38   54.21  702.19   57.23   700.5   63.25  698.79
   72.29  694.89   81.32  691.67   84.33  691.06   99.39  689.62  114.31  689.02
  117.25  689.07  120.71  689.66  126.41  691.18  136.62  691.99  139.65  692.61
  148.73   696.1   157.8  700.96  163.85  702.89  191.09  708.94  200.16  710.53
  206.22  712.09  218.32  713.12  230.42  715.01  245.55  718.94  248.58  719.24
#Mann= 3 , 0 , 0
       0      .1       0   99.39      .1       0  120.71      .1       0
Bank Sta=99.39,120.71
XS Rating Curve= 0 ,0
Exp/Cntr=0.3,0.1

Type RM Length L Ch R = 1 ,5394.959,79.64,91.44,94.03
XS GIS Cut Line= 3
     625971.8838    4341822.9451     625898.9482    4341947.3283
     625861.8169    4342050.4872
#Sta/Elev= 30
       0  719.42    3.07  719.23     9.2   716.9   15.34  713.47   24.54  707.12
   27.61   705.7   33.75  703.83   39.88  700.91   42.95  700.14   46.02  697.96
   49.09  696.63   55.22   691.6   58.29  689.71   61.36  688.68    76.7  689.09
  138.05  688.63  147.24  687.73  150.32  688.84  153.33  690.71  156.37  691.52
  159.42  694.95  162.46  697.33  174.65  702.85  183.78  705.79  189.87   706.8
   205.1  711.44  217.28  714.18  223.37  714.84  250.78  719.91  253.83  720.07
#Mann= 3 , 0 , 0
       0      .1       0  138.05      .1       0  150.32      .1       0
Bank Sta=138.05,150.32
XS Rating Curve= 0 ,0
Exp/Cntr=0.3,0.1

Type RM Length L Ch R = 1 ,5303.52 ,87.25,91.44,80.62
XS GIS Cut Line= 4
     625935.9004    4341792.2534     625850.6152    4341872.4145
     625832.2115    4341886.9116       625751.75    4341965.8204
#Sta/Elev= 30
       0  720.23       9  715.89   15.01  713.55   18.01  712.85   30.01  707.02
   36.01  705.28   45.02  701.82   51.02  700.06   57.02  697.81   60.02  696.08
   63.02  693.12   69.03  691.08   78.03  686.84   81.03  686.15  126.66  686.02
  134.62  685.68  140.47  686.08  149.61  687.02  152.66   688.1  158.75  691.27
  164.84  693.91  167.88  694.93  173.98  696.04  180.07  698.04  189.21  702.55
   195.3  705.09  198.34  706.04   228.8  712.62  244.03  716.57  253.17  719.65
#Mann= 3 , 0 , 0
       0      .1       0  126.66      .1       0  140.47      .1       0
Bank Sta=126.66,140.47
XS Rating Curve= 0 ,0
Exp/Cntr=0.3,0.1

Type RM Length L Ch R = 1 ,5212.08 ,97.5,91.86,87.59
XS GIS Cut Line= 6
     625872.4003    4341724.5199     625806.9049    4341796.9778
      625805.769    4341805.7856     625792.0994    4341821.8983
     625785.7382    4341823.4362     625688.2499    4341927.7203
#Sta/Elev= 30
       0   720.5   12.21  715.61   15.26  713.62   36.63  703.24   42.73  701.41
   45.78  700.11   48.84  699.48   67.15   691.5   82.41   685.4   91.57  683.79
   97.67  683.22  106.55  683.88  158.53  684.04  161.56  684.48   164.6  685.62
  173.71  691.66  176.75  692.67  179.79  693.09  182.82  694.04   188.9  696.03
  194.97  698.62  210.16  703.43  222.31     707  228.39  708.15  240.53  711.35
  255.72  714.43  267.87  717.64  270.91  718.07  273.95  719.07  276.98  719.48
#Mann= 3 , 0 , 0
       0      .1       0   91.57      .1       0  106.55      .1       0
Bank Sta=91.57,106.55
XS Rating Curve= 0 ,0
Exp/Cntr=0.3,0.1

Type RM Length L Ch R = 1 ,5120.215,100.89,91.02,97.47
XS GIS Cut Line= 2
     625821.6002    4341656.7864     625624.7498    4341887.5036
#Sta/Elev= 30
       0  720.52   12.25  715.44   15.32  714.67   21.44   712.2   45.95   703.7
   55.14  699.94   58.21  699.29   61.27  699.07   85.78  690.96    91.9  686.96
   98.03  681.78  101.09  680.38  104.16  680.21  110.28  680.87  113.35   681.2
  165.43  682.52  171.55  683.13  174.62  684.17  189.93  691.03     193  691.56
  202.19  695.36  220.57  701.34   226.7  703.61  229.76  705.25  232.82  706.46
  238.95  708.58  263.46   713.9  278.78  716.28   284.9  716.84  303.28  717.16
#Mann= 3 , 0 , 0
       0      .1       0  101.09      .1       0  110.28      .1       0
Bank Sta=101.09,110.28
XS Rating Curve= 0 ,0
Exp/Cntr=0.3,0.1

Type RM Length L Ch R = 1 ,5029.2  ,86,91.44,87.32
XS GIS Cut Line= 6
     625736.9333     4341589.053     625694.7214    4341664.5006
      625693.353    4341670.3276     625685.2587    4341681.7256
     625664.9557    4341687.9163     625540.0829      4341749.92
#Sta/Elev= 30
       0  709.71    8.94  706.33   26.83  697.97   29.81  697.17   38.75  695.55
   41.74  694.22    47.7  690.87   59.62  685.22   65.59  681.63   68.57  680.12
   71.55  679.42   80.49  679.18   95.23  678.59  106.42  679.17  127.64  679.06
  136.74  679.36   142.8  679.92  145.83  680.98  148.86  682.76  167.05  688.81
  173.11  691.42  191.29  696.85  197.35  699.17  224.63  705.19  230.69  705.99
  239.79  707.72  245.85  709.33  248.88  709.87  254.94  710.51  267.06  711.02
#Mann= 3 , 0 , 0
       0      .1       0   80.49      .1       0  127.64      .1       0
Bank Sta=80.49,127.64
XS Rating Curve= 0 ,0
Exp/Cntr=0.3,0.1

Type RM Length L Ch R = 1 ,4937.76 ,90.28,91.71,93.51
XS GIS Cut Line= 4
      625716.137    4341539.0995     625629.3394    4341607.9298
     625620.8266    4341615.6318     625533.5742    4341724.0437
#Sta/Elev= 30
       0  710.82    8.98  707.26   14.97  703.72   32.93  695.72   38.92  694.13
   44.91  692.09   62.87  685.25   68.86  682.47   71.86  679.93   74.85   678.2
   77.84  677.51   80.84  677.35  107.78  677.26  116.52  677.04  119.39  677.15
  122.26  677.83  131.33  681.09  137.38  682.77  152.51  685.74  164.61  688.93
  170.66  690.91  188.81  695.57  197.89  697.37  203.94  699.15  209.99  701.96
  216.04  703.91  222.09   705.1  237.22  706.84  255.37   710.6  261.42  711.12
#Mann= 3 , 0 , 0
       0      .1       0  107.78      .1       0  119.39      .1       0
Bank Sta=107.78,119.39
XS Rating Curve= 0 ,0
Exp/Cntr=0.3,0.1

Type RM Length L Ch R = 1 ,4846.053,84.12,91.3,92.57
XS GIS Cut Line= 2
      625687.562    4341461.3119     625484.1166    4341597.4705
#Sta/Elev= 30
       0  712.21   12.24   707.4    15.3  705.23   21.42  702.63   27.54  700.54
   36.72  698.15   42.84  695.24   55.08  690.04   64.26  688.15   73.44  684.17
   79.56  681.96    91.8  675.75   94.86  674.94   97.92  674.72  119.34  674.45
  125.46  674.19  146.88  674.09  151.21  674.43  171.36  677.32  174.42  678.21
  177.48  679.48  180.54  681.37  189.72  689.34  192.78  691.15  195.84   692.6
  201.96  696.65   214.2  701.59  223.38  704.77  226.44  706.32   244.8  711.05
#Mann= 3 , 0 , 0
       0      .1       0  119.34      .1       0  151.21      .1       0
Bank Sta=119.34,151.21
XS Rating Curve= 0 ,0
Exp/Cntr=0.3,0.1

Type RM Length L Ch R = 1 ,4754.749,104.98,91.31,85.1
XS GIS Cut Line= 2
     625668.5119    4341428.7681      625428.799    4341485.1244
#Sta/Elev= 30
       0  711.38    6.08  708.98    9.12  706.97   12.16  705.51   27.36  699.51
   33.44  696.25   54.72  688.91   69.92  681.04   72.96  678.11   82.08  674.04
   85.12  673.22   88.16  672.92   97.28  672.67  139.84  672.82  148.97  672.19
  150.01  672.47  152.01  672.99  155.05  675.09  158.09  678.78  176.33  688.39
  179.37  690.96  182.41  692.96  185.45  694.35  197.61  698.33  203.69   700.8
  215.85  703.41  221.93  705.73  231.05  707.59  243.21  710.97  246.25  711.52
#Mann= 3 , 0 , 0
       0      .1       0   97.28      .1       0  150.01      .1       0
Bank Sta=97.28,150.01
XS Rating Curve= 0 ,0
Exp/Cntr=0.3,0.1

Type RM Length L Ch R = 1 ,4663.44 ,86.41,91.71,92.36
XS GIS Cut Line= 5
     625727.6464    4341131.3758     625520.1566    4341372.5048
     625516.6463    4341381.3045     625507.2943    4341395.9045
     625435.9427    4341433.0014
#Sta/Elev= 30
       0  702.92   12.24  697.15   27.53  696.08   55.06  697.13   61.18  696.44
    88.7  699.07  137.64  700.18  162.11  698.28  168.23  697.11  189.64  696.08
  195.76  695.11  198.82  693.59  201.88  693.14  214.11  687.68  238.58  681.44
  250.82  678.81  256.94  678.15     260   677.2  272.23  671.35  275.29  670.65
  308.94  669.55  333.37     669  336.26  669.17  339.14  670.47   347.9  676.07
  350.88  678.53   362.8  684.08  374.71  688.24  395.56   693.1  425.34  701.97
#Mann= 3 , 0 , 0
       0      .1       0  308.94      .1       0  336.26      .1       0
Bank Sta=308.94,336.26
XS Rating Curve= 0 ,0
Exp/Cntr=0.3,0.1

Type RM Length L Ch R = 1 ,4571.733,83.83,90.98,92.34
XS GIS Cut Line= 3
     625662.8234     4341144.605     625498.9739    4341274.4174
     625379.7187    4341387.3607
#Sta/Elev= 30
       0  700.86    9.22  698.31   15.37  698.22   18.44  697.34   33.82  695.11
   46.11  691.82   67.63  684.66  113.74   681.5  122.96  680.54  132.19  678.78
  162.93  676.83  181.37  674.95  187.52  674.84  193.67  675.42  209.04   675.2
  215.12  673.89  224.25  669.95  227.29   669.2  245.54     668  269.87  667.14
  272.92  667.46     279  672.49  282.04  673.95  291.17  677.66  297.25  679.14
  306.37  683.46  336.79  692.19  345.92  693.83  358.08  697.02  373.29  701.78
#Mann= 3 , 0 , 0
       0      .1       0  245.54      .1       0  272.92      .1       0
Bank Sta=245.54,272.92
XS Rating Curve= 0 ,0
Exp/Cntr=0.3,0.1

Type RM Length L Ch R = 1 ,4480.751,57.67,91.63,101.82
XS GIS Cut Line= 2
     625589.4014    4341169.7405     625314.2342    4341280.8657
#Sta/Elev= 30
       0  692.82    15.3  690.46   18.36  689.61   27.53  685.64   30.59  684.94
   64.25  682.35   79.54  679.68   91.78  678.13  128.49  675.25  137.67  674.24
  140.73  673.64  143.79  672.64  152.97  668.26  156.03  667.03  159.09  666.55
  186.62  666.08  198.86  665.97  208.04  665.57   211.1  665.58  214.16  665.97
  223.33  667.05  229.45  670.06  244.75   674.6  250.87  676.91  269.22  682.51
  272.28  683.98  275.34  685.11  290.64  690.03   293.7  691.24  296.76  693.09
#Mann= 3 , 0 , 0
       0      .1       0  186.62      .1       0  214.16      .1       0
Bank Sta=186.62,214.16
XS Rating Curve= 0 ,0
Exp/Cntr=0.3,0.1

Type RM Length L Ch R = 1 ,4389.12 ,124.23,91.44,61.89
XS GIS Cut Line= 6
     625502.0887    4341141.2977     625373.6673    4341202.8991
     625357.0373    4341187.2642      625356.743    4341181.2272
     625345.0816    4341176.0239     625258.0101     4341186.277
#Sta/Elev= 30
       0  693.46    3.03  692.79    9.09  690.09    30.3  683.95   33.34  682.53
   45.46  678.14   57.58  674.31   63.64  673.36   78.79  672.29   90.91  669.43
   96.97  666.36  100.01  665.17  106.07  664.51   139.4  663.62  159.55  663.56
   171.3  663.05  177.56  663.66     188  664.07  197.07  663.73  200.09   664.1
  212.18  671.06  218.23  675.13  221.25  678.17  224.28  679.79  233.35  682.22
  239.39  682.82  242.42  683.61  257.53  687.82   266.6  691.09  272.65  692.77
#Mann= 3 , 0 , 0
       0      .1       0   139.4      .1       0  177.56      .1       0
Bank Sta=139.4,177.56
XS Rating Curve= 0 ,0
Exp/Cntr=0.3,0.1

Type RM Length L Ch R = 1 ,4297.68 ,41.49,91.44,104.43
XS GIS Cut Line= 6
     625471.3639    4341057.5238     625353.3365    4341082.1075
     625349.3678    4341094.8075     625344.6207    4341116.7894
     625331.5083    4341126.5575     625240.1176    4341157.5365
#Sta/Elev= 30
       0  692.91    6.03  691.27    9.04  689.69   27.13   684.5   33.15  682.21
   45.21  679.02   51.24  676.26   69.32   670.7   72.34   669.2   78.36  668.33
   81.38  667.38   90.42  664.06   93.43  662.32   96.45  661.56  125.88  661.39
  136.47  661.97  142.21  661.03  147.32  660.68  153.41  661.25  161.91  662.08
  170.09  662.03  190.91  662.79  193.92   663.9  202.97  668.85  215.03  674.05
  224.08  676.83  233.12  679.21  236.14  680.68  254.23   686.4  269.31     693
#Mann= 3 , 0 , 0
       0      .1       0  142.21      .1       0  153.41      .1       0
Bank Sta=142.21,153.41
XS Rating Curve= 0 ,0
Exp/Cntr=0.3,0.1

Type RM Length L Ch R = 1 ,4206.24 ,108.09,91.44,77.73
XS GIS Cut Line= 5
     625470.6583    4341045.1766     625357.7604    4341065.2958
      625342.833    4341052.9215     625325.8842    4341035.7872
     625200.9592    4341017.8363
#Sta/Elev= 30
       0  692.84    3.02  691.83    6.04   690.3   24.14  685.38   27.16  683.82
   45.27  679.27    51.3  676.79   63.37   672.9   69.41  669.97   81.48  667.62
   87.52  665.48   90.53  663.84   96.57  662.05  102.61  661.38  128.53  660.79
  140.09  658.83  146.12  658.49  155.15  659.16  161.17  659.38  194.23  659.17
  200.24  660.49  215.26  665.99  221.27  669.66  233.29  674.31   239.3  677.77
  254.33  683.65  257.33  685.05  260.34  686.94  272.35  690.46  284.37  692.91
#Mann= 3 , 0 , 0
       0      .1       0  140.09      .1       0  155.15      .1       0
Bank Sta=140.09,155.15
XS Rating Curve= 0 ,0
Exp/Cntr=0.3,0.1

Type RM Length L Ch R = 1 ,4114.8  ,92.96,91.44,88.95
XS GIS Cut Line= 3
     625467.4833    4340930.8764     625324.7466    4340958.0021
     625178.5578    4340958.3931
#Sta/Elev= 30
       0  693.84    6.05  691.06   12.11  687.77   18.16  685.67   27.24  683.09
   30.27  681.66   48.43  677.58   66.59  671.98   75.67  668.54   81.73  666.76
   90.81  664.73   93.83  663.01  108.97  658.54  115.02  657.46   124.1     657
  130.16  656.73  151.38  656.92  194.02  657.26  197.07  657.71  200.11  658.84
  212.29  664.68  218.39  668.64  230.57  673.15  236.66  677.15  242.75  679.75
  251.89  681.99  257.98  683.85  270.16  686.43  276.25  688.43  291.48  691.41
#Mann= 3 , 0 , 0
       0      .1       0   124.1      .1       0  151.38      .1       0
Bank Sta=124.1,151.38
XS Rating Curve= 0 ,0
Exp/Cntr=0.3,0.1

Type RM Length L Ch R = 1 ,4023.36 ,81.44,91.44,102.35
XS GIS Cut Line= 4
     625445.8404    4340846.2095     625343.4436     4340858.669
     625303.4296    4340870.5898     625218.8274    4340878.7533
#Sta/Elev= 30
       0  683.59     9.1  679.77    18.2  676.64   36.41   673.1   39.44  671.29
   54.61  665.92   57.64  663.63   60.68  662.59   63.71  662.03   72.81  661.36
   75.85  660.59   78.88  658.19   81.91  656.55   84.95  655.75  129.99  655.11
  138.94  654.38  141.92  655.02   144.9  655.35  163.12  655.33  166.15  655.55
  169.19  656.31  178.29  660.52  184.37  665.44  190.44  668.53  202.58  673.13
  205.61  674.78  220.79  679.94  223.83  681.17  226.86  682.94   229.9  683.86
#Mann= 3 , 0 , 0
       0      .1       0  129.99      .1       0  141.92      .1       0
Bank Sta=129.99,141.92
XS Rating Curve= 0 ,0
Exp/Cntr=0.3,0.1

Type RM Length L Ch R = 1 ,3931.917,92.02,91.46,91.55
XS GIS Cut Line= 4
     625451.3966    4340792.2344     625327.8596    4340782.0222
     625317.0166     4340780.222     625240.2587    4340755.7218
#Sta/Elev= 30
       0  684.96   12.09  680.15   18.14   676.4   30.23  671.53   36.28  668.84
    51.4  664.81   54.42  663.86   57.44   662.4   63.49  660.47   66.51  659.66
   72.56   658.8   75.58  657.19   81.63  655.33   87.68  654.13   99.77  652.65
  129.45  651.57  140.92  651.14   143.9   651.2  146.89   651.9  149.87  653.45
  152.85  655.27  155.84     658  158.82  660.09  164.79  663.08  173.74  666.75
  176.73  668.48  185.68  671.19   200.6  675.28  206.57  677.92  215.52  682.94
#Mann= 3 , 0 , 0
       0      .1       0  129.45      .1       0   143.9      .1       0
Bank Sta=129.45,143.9
XS Rating Curve= 0 ,0
Exp/Cntr=0.3,0.1

Type RM Length L Ch R = 1 ,3840.457,85.22,91.42,92.99
XS GIS Cut Line= 3
     625447.2956    4340714.9098     625333.9826    4340690.3431
     625241.5816     4340677.868
#Sta/Elev= 30
       0  685.02    3.05   682.6     6.1  681.01   18.31  675.78   24.41     672
   39.67  666.04   45.77  662.76   57.97  658.78   64.08  656.15   82.38  653.38
   88.48  652.97   91.54  652.31   97.64     650  100.69  649.18  103.74  648.83
  118.95  648.51  124.97  649.26  130.98  650.11     137  651.83  146.02  656.59
  158.05  661.61  161.06  663.22  164.07  665.47  179.11  670.76  182.12  672.53
  191.14  673.63  194.15  674.59  200.16  677.75  203.17  680.95  209.18  684.99
#Mann= 3 , 0 , 0
       0      .1       0  100.69      .1       0  124.97      .1       0
Bank Sta=100.69,124.97
XS Rating Curve= 0 ,0
Exp/Cntr=0.3,0.1

Type RM Length L Ch R = 1 ,3749.04 ,12.83,13.36,19.54
XS GIS Cut Line= 6
     625437.3737    4340627.5971     625357.8305    4340614.0273
     625351.2159    4340614.1596      625341.824    4340601.4148
     625331.5242    4340596.6384     625239.5973    4340592.5398
#Sta/Elev= 30
       0  683.84    2.99  680.67    5.98  679.11   17.93  675.28   20.92  672.97
   23.91   671.4   38.85  665.21   44.83  661.21   50.81  658.43   56.78  655.06
   59.77  652.78   62.76   649.6   65.75  648.46   68.74  648.03    85.1  648.71
      98  648.07  103.16  647.26  105.77  647.31  108.39  648.13  110.45   648.6
  123.77  649.79  142.17  656.04  151.37  659.77  163.64  663.97  169.78  667.21
  178.98  670.74  182.05  672.21  188.18  677.07  191.25  678.44  206.58  683.23
#Mann= 3 , 0 , 0
       0      .1       0      98      .1       0  108.39      .1       0
Bank Sta=98,108.39
XS Rating Curve= 0 ,0
Exp/Cntr=0.3,0.1

Type RM Length L Ch R = 1 ,3735.676,90.33,78.14,66.55
XS GIS Cut Line= 6
     625435.3893    4340622.9669     625357.8159    4340611.7809
     625355.7522    4340602.4147     625347.5765    4340594.9534
     625337.9721    4340575.9034     625237.6129    4340581.2949
#Sta/Elev= 30
       0  681.97    6.03  678.43   15.07  675.73    21.1  672.02   36.17  665.44
    42.2  661.48   54.26  655.47   57.27  653.31   60.29  649.83    63.3  648.46
   66.32  647.87   78.38  648.55   96.49  647.62  106.02   646.9  110.77  647.64
  119.51   648.6  137.05  648.99  149.34  651.33  155.49  653.14  158.56  654.15
  161.63  655.96  176.99  661.26  180.07  663.37  192.36  668.21   198.5  671.51
  201.57  675.24  204.65  676.86  216.94  680.89  220.01  682.78  223.08  683.71
#Mann= 3 , 0 , 0
       0      .1       0   96.49      .1       0  110.77      .1       0
Bank Sta=96.49,110.77
XS Rating Curve= 0 ,0
Exp/Cntr=0.3,0.1

Type RM Length L Ch R = 1 ,3657.534,92.44,91.33,93.71
XS GIS Cut Line= 3
     625446.3695    4340511.3897     625345.4033    4340512.6675
     625239.9941    4340504.2459
#Sta/Elev= 30
       0   684.1    15.3  676.92   18.36  674.22   36.72  666.81   39.78  664.35
   55.08   657.9   58.14  655.68    76.5  649.99   79.56  648.27   88.74  645.42
   91.79  644.72   94.85  644.69   97.91  645.34  116.08  645.73   119.1  646.15
  122.12     647  134.21  651.69  137.23  653.74  140.25  655.21  143.27  656.23
  146.29  656.82  152.34  656.86  155.36  657.32   161.4  660.87  173.49     666
  179.53  669.89  185.57  672.67  191.61  675.84  197.66  679.71  206.72  683.48
#Mann= 3 , 0 , 0
       0      .1       0   88.74      .1       0   97.91      .1       0
Bank Sta=88.74,97.91
XS Rating Curve= 0 ,0
Exp/Cntr=0.3,0.1

Type RM Length L Ch R = 1 ,3566.207,98,91.49,86.77
XS GIS Cut Line= 4
      625441.607    4340437.5708      625347.398    4340421.3298
     625339.7814    4340418.5977     625250.3129     4340405.027
#Sta/Elev= 30
       0  675.76    2.99  673.59    5.97  671.89   17.92  667.27    23.9  663.87
   32.86   660.8   41.82  658.19   44.81  656.67   59.75     652    71.7   644.5
   74.69  643.66   80.66  643.17   89.62  640.59   92.61  640.16    95.6  640.26
   97.85  640.71  103.69  642.12  112.74  643.19  115.76  644.14  118.77  645.64
  124.81  650.97  127.82  652.29  139.89  656.34  145.92  659.46  154.97  662.59
  157.99  663.45  167.03  664.34  182.12  670.08  185.13   672.2  194.18  675.28
#Mann= 3 , 0 , 0
       0      .1       0   89.62      .1       0   97.85      .1       0
Bank Sta=89.62,97.85
XS Rating Curve= 0 ,0
Exp/Cntr=0.3,0.1

Type RM Length L Ch R = 1 ,3474.72 ,93.2,91.44,79.51
XS GIS Cut Line= 6
     625425.4145    4340310.6764     625366.9233    4340333.0049
     625361.9624    4340333.0049     625355.3803    4340333.5769
     625328.5628    4340333.2458     625228.5641    4340360.6827
#Sta/Elev= 30
       0   675.3    8.94  671.16   14.91     667   23.85     663   32.79  658.62
   35.78  655.87    47.7  648.97   53.66  645.12   56.65  642.72   59.63  639.34
   62.61  638.85   65.09  638.95   67.57  639.46   71.97  640.65   74.18  640.84
   95.04  640.69   98.02  641.52  104.05  644.39  119.29  650.58  122.34  652.47
  131.49  655.78  140.64  658.66  143.69  660.79  146.74  662.13  155.89  665.35
  165.04  667.91  171.14  668.68  183.34  669.42  198.59  672.73  204.69  674.34
#Mann= 3 , 0 , 0
       0      .1       0   59.63      .1       0   67.57      .1       0
Bank Sta=59.63,67.57
XS Rating Curve= 0 ,0
Exp/Cntr=0.3,0.1

Type RM Length L Ch R = 1 ,3383.28 ,98.24,91.62,87.06
XS GIS Cut Line= 4
     625380.1707    4340220.9824     625350.4598    4340242.6041
     625345.2294    4340250.4945     625226.9766    4340355.1264
#Sta/Elev= 30
       0   675.1    6.12   668.3   18.37  653.81   21.43  649.49    24.5  645.49
   27.56  643.13   30.62  640.03   33.68   638.3   36.75  637.76   39.11  637.94
   41.48  638.36   46.21   639.1   58.36  639.82   61.39  640.34    70.5  642.88
   88.72  646.18  103.91  648.73  109.98  650.12  116.05  652.19  125.16  654.62
   128.2  655.37  131.23  655.82  140.34  658.08  146.42  660.42  164.64  666.75
  173.74  669.44  185.89  670.35  191.96  671.03  198.04  672.45  204.11  674.52
#Mann= 3 , 0 , 0
       0      .1       0   33.68      .1       0   41.48      .1       0
Bank Sta=33.68,41.48
XS Rating Curve= 0 ,0
Exp/Cntr=0.3,0.1

Type RM Length L Ch R = 1 ,3291.656,81.45,91.26,99.98
XS GIS Cut Line= 3
     625330.1643    4340165.4198     625277.6856    4340193.9319
     625211.8953    4340286.8638
#Sta/Elev= 30
       0  666.38   14.93  661.77    20.9  659.66   23.89  657.71   29.86  655.01
   32.85  653.75   35.83  652.88   38.82  651.24   44.79  649.73   50.77  646.72
   59.72  643.04   71.71   637.4   78.27  634.95    80.7  634.46    83.7  634.38
   89.69  634.96   92.68  634.99   95.68  635.43   98.68  636.79  104.67  640.55
  110.66  643.69  113.66  645.07  119.65  647.37  128.64  652.09  131.64  653.37
  134.63  653.82  146.62   658.2   161.6  662.65  167.59  664.76  173.59  665.97
#Mann= 3 , 0 , 0
       0      .1       0   78.27      .1       0   89.69      .1       0
Bank Sta=78.27,89.69
XS Rating Curve= 0 ,0
Exp/Cntr=0.3,0.1

Type RM Length L Ch R = 1 ,3200.4  ,88.6,91.42,95.53
XS GIS Cut Line= 5
     625331.2888    4340154.8629     625268.6794    4340144.6815
     625247.0764    4340132.5206     625227.9273    4340131.8714
     625159.9707    4340114.5139
#Sta/Elev= 30
       0  666.56    3.02  665.18    15.1  661.48   21.14  658.44   36.25  653.08
   39.27   651.4   42.29  650.13   57.39  645.42   60.41  643.18    71.7   637.6
    77.2  635.14   82.71  632.01   88.22  629.89    93.7  629.33   96.43  629.43
   99.17  629.91  119.58  632.81  122.63   633.6  128.73   634.1  131.78  634.93
  134.83  636.64  137.88  638.69  140.93  642.27  143.98  644.64  156.17  651.06
  159.22  653.42  162.27  656.71  165.32  659.23  168.37  661.14  177.52  665.82
#Mann= 3 , 0 , 0
       0      .1       0   88.22      .1       0   99.17      .1       0
Bank Sta=88.22,99.17
XS Rating Curve= 0 ,0
Exp/Cntr=0.3,0.1

Type RM Length L Ch R = 1 ,3108.978,96.15,91.52,83.63
XS GIS Cut Line= 4
     625354.4399    4340117.1597     625272.2453    4340053.2714
     625253.4554    4340037.0816      625164.601    4340051.0138
#Sta/Elev= 30
       0  666.03    3.06  665.32   18.37  658.31    24.5  654.75    39.8  647.62
   42.87  646.67   55.11  640.31    64.3  635.22   70.42  631.43   73.49  630.38
   76.55  629.82   88.79  629.42   94.92  627.84   97.98  627.43  101.04  627.36
  106.86  628.07  109.62  628.74  117.88   632.4   123.4  633.85  128.91   635.8
   134.9  637.47   137.9  639.34  152.89  645.78  161.88  650.21  179.87  657.06
  188.87  658.59  197.86  660.84  200.86  661.89  209.85  663.65  218.85  665.91
#Mann= 3 , 0 , 0
       0      .1       0   94.92      .1       0  106.86      .1       0
Bank Sta=94.92,106.86
XS Rating Curve= 0 ,0
Exp/Cntr=0.3,0.1

Type RM Length L Ch R = 1 ,3017.46 ,95.28,91.42,67.63
XS GIS Cut Line= 4
     625457.6276    4339963.7011     625307.4397    4339978.6793
     625284.9376      4339979.34     625181.7989    4340036.4616
#Sta/Elev= 30
       0  655.62    9.06   655.5   24.15   654.2   39.24  653.34   51.32  651.75
   60.37  650.13    81.5  645.14   84.52     644   90.56   642.4  102.63  639.94
  120.75  632.01  126.78  627.51   129.8  625.98  132.82  625.13  135.84  624.98
  141.88   625.5  147.91  626.71  150.93  626.94  167.82  627.64  185.54  627.75
  197.63  629.75  203.68  630.22   206.7  630.81  218.79  634.47  239.95  642.29
     246  643.94  249.02  645.78  255.07  646.78  270.18  651.29  291.35  655.93
#Mann= 3 , 0 , 0
       0      .1       0  132.82      .1       0  141.88      .1       0
Bank Sta=132.82,141.88
XS Rating Curve= 0 ,0
Exp/Cntr=0.3,0.1

Type RM Length L Ch R = 1 ,2926.037,94.15,91.34,79.53
XS GIS Cut Line= 4
     625270.5668    4339879.1665      625244.026    4339937.8512
     625234.7827    4339963.3877      625168.702    4340035.9325
#Sta/Elev= 30
       0   657.7    6.13  652.34   12.27  647.82   15.34  646.75   21.47  641.01
    36.8  627.22   39.87     625   42.94  623.99   50.25  623.55   55.21  622.55
   58.27  622.54   61.34  623.27   67.42  624.92   70.44  625.35   91.57  627.36
  103.83  628.29   106.9  628.97  113.03  631.47   116.1  632.25  119.16  632.82
   125.3  632.65  128.36  633.19  131.43  634.16   134.5  635.45  140.63  638.55
  146.76  641.05  165.16  647.81   171.3  648.55  183.56  653.57  189.69  656.36
#Mann= 3 , 0 , 0
       0      .1       0   50.25      .1       0   61.34      .1       0
Bank Sta=50.25,61.34
XS Rating Curve= 0 ,0
Exp/Cntr=0.3,0.1

Type RM Length L Ch R = 1 ,2834.698,91.36,91.56,88.8
XS GIS Cut Line= 3
     625131.6603    4339832.8644     625166.7401    4339960.5795
      625152.827    4340031.3023
#Sta/Elev= 30
       0  657.02    6.02  653.74   12.04  651.15   18.06  649.88   42.14  639.75
   45.15  639.34   48.16  638.07   57.19  633.41   66.22  627.74   69.23  626.29
   72.24  625.36   78.26  624.73   93.31  622.05  102.34  620.81  108.36  620.43
  117.39   619.2   120.4  619.37  123.41  620.45  132.45  624.63  135.45  625.43
  138.45  625.44  150.46  628.02  165.48   635.6  168.48  636.02  171.49  637.03
   186.5  645.39  195.51  652.18  198.52     654  201.52  654.71  204.52  656.85
#Mann= 3 , 0 , 0
       0      .1       0  108.36      .1       0   120.4      .1       0
Bank Sta=108.36,120.4
XS Rating Curve= 0 ,0
Exp/Cntr=0.3,0.1

Type RM Length L Ch R = 1 ,2743.138,85.89,91.28,75.2
XS GIS Cut Line= 3
     625039.7174    4339854.6925     625073.3268    4339949.0125
     625101.8946    4340046.5158
#Sta/Elev= 30
       0  656.61    3.03  654.62    6.07  653.81     9.1  652.62   21.24  644.08
   33.38  636.06   39.44  633.65   48.55  626.28   51.58  624.37   54.62  622.82
   57.65   621.6   60.68  620.78   66.75  619.85   69.79  619.77   78.89  618.13
   87.99  617.73   97.09  617.81  106.11  618.39  115.07  618.16  118.06   618.9
  124.04  621.05  135.99  622.06  141.97  623.28  144.95  624.32  150.93  627.37
  156.91  631.07   159.9  631.64   183.8  646.21  189.78  648.34  201.73  656.86
#Mann= 3 , 0 , 0
       0      .1       0   78.89      .1       0  106.11      .1       0
Bank Sta=78.89,106.11
XS Rating Curve= 0 ,0
Exp/Cntr=0.3,0.1

Type RM Length L Ch R = 1 ,2651.859,89.69,91.36,102.35
XS GIS Cut Line= 2
     624959.5705    4339908.3259     625062.7582    4340059.1387
#Sta/Elev= 30
       0  647.73    3.05  644.79    9.14  640.98   15.23  636.84   24.36  629.72
   30.46  627.31    33.5  624.82   36.55  622.68   39.59  620.79   45.68  616.42
   48.73  614.73   51.78  614.41   54.82  615.44   57.87  616.61   60.91   617.1
   63.96  617.26   76.14  617.33   88.32  617.95  121.82  620.67  124.87   621.1
  130.96  621.51  134.01     622  137.05   623.2  149.23  629.42  155.33  633.35
  158.37  633.97  161.42  635.08  167.51  638.13  176.64   643.2  182.74     647
#Mann= 3 , 0 , 0
       0      .1       0   48.73      .1       0   54.82      .1       0
Bank Sta=48.73,54.82
XS Rating Curve= 0 ,0
Exp/Cntr=0.3,0.1

Type RM Length L Ch R = 1 ,2560.497,94.08,91.72,82.54
XS GIS Cut Line= 2
     624904.6694    4339936.1072     624937.0809    4340186.8004
#Sta/Elev= 30
       0  646.62    3.05  644.97    6.09  644.56   21.32  634.38   30.46  627.21
    33.5  627.06   36.55  624.46   42.64  617.73   45.68  615.32   54.82   613.5
   60.91  613.58   63.96  613.63   73.09  614.85   76.14  614.82  118.78  612.73
  130.96   612.8     134  613.15  143.14  614.74  149.23  616.52  170.55  618.91
  179.69  620.92  182.73  621.11  188.82   622.7  201.01  626.16  210.14  629.66
  213.19   629.8  222.32  634.37  237.55  640.96  243.64  642.83  252.78   648.1
#Mann= 3 , 0 , 0
       0      .1       0   54.82      .1       0   60.91      .1       0
Bank Sta=54.82,60.91
XS Rating Curve= 0 ,0
Exp/Cntr=0.3,0.1
